--- ArmstrngCk.prj (project) ---

Proj Title=ArmstrngCk
Current Plan=p01
Default Exp/Contr=0,0
English Units
Geom File=g01
Flow File=f01
Plan File=p01
BEGIN DESCRIPTION:
END DESCRIPTION:
DSS Export Rating Curves= 0
DSS Export Rating Curve Sorted= 0
DSS Export Volume Flow Curves= 0
DXF OffsetX= 0
DXF OffsetY= 0
DXF ScaleX= 0
DXF ScaleY= 0

--- ArmstrngCk.p01 (plan) ---

Plan Title=Floodplain
Program Version=4.00
Geom File=g01
Flow File=f01
K Sum by GR=0
Std Step Tol=0.01
Critical Tol=0.01
Num of Std Step Trials=20
Max Error Tol=0.3
Flow Tol Ratio=0.001
Split Flow NTrial=30
Split Flow Tol=0.02
Split Flow Ratio=0.02
Log Output Level=0
Friction Slope Method=1
Unsteady Friction Slope Method=2
Unsteady Bridges Friction Slope Method=1
Global Log Level=0
CheckData=False
Run HTab=0
Run UNet=0
Run PostProcess=0
UNET Theta=0
UNET Theta Warmup=0
UNET ZTol=0
UNET ZSATol=0
UNET MxIter=0
UNET MaxInSteps=0
UNET DtIC=0
UNET DtMin=0
UNET MaxCRTS=0
UNET WFStab=0
UNET SFStab=0
UNET WFX=0
UNET SFX=0
UNET DSS MLevel=0
UNET DZMax Abort=0
UNET Convert EG Bridges=0
UNET Use Existing IB Tables=0
UNET Froude Limit=0
UNET Froude Power=0
Write IC File=0
Echo Input=False
Echo Output=False
Write Detailed=0

--- ArmstrngCk.f01 (steady flow) ---

Flow Title=NFF Regression Equation
Program Version=4.10
Number of Profiles= 1
Profile Names=P100yr
River Rch & RM=ArmstrngCk,Main            ,40107.8
930.1523
River Rch & RM=ArmstrngCk,Main            ,39807.8
1374.567
River Rch & RM=ArmstrngCk,Main            ,38007.8
1491.052
River Rch & RM=ArmstrngCk,Main            ,36175.3
1625.726
River Rch & RM=ArmstrngCk,Main            ,32907.8
1746.572
River Rch & RM=ArmstrngCk,Main            ,29155.2
1936.086
River Rch & RM=ArmstrngCk,Main            ,25103.9
2150.341
River Rch & RM=ArmstrngCk,Main            ,18318.4
  2382.7
River Rch & RM=ArmstrngCk,Main            ,17607.8
3446.414
River Rch & RM=ArmstrngCk,Main            ,14746.2
3803.024
River Rch & RM=ArmstrngCk,Main            ,5940.3
4193.755
River Rch & RM=ArmstrngCk,Main            ,57.8
4521.351
Boundary for River Rch & Prof#=ArmstrngCk,Main            , 1
Up Type= 0
Dn Type= 3
Dn Slope=0.007624
DSS Import GetInterval= 0
DSS Import GetPeak= 0
DSS Import FillOption= 0

--- ArmstrngCk.g01 (geometry) ---

Geom Title=USGS 3m DEM
Program Version=4.10

River Reach=ArmstrngCk      ,Main
Reach XY= 30
     1873880.094      381018.362     1873084.387      381825.173
     1871740.637      385872.049     1871781.663      386451.411
      1871315.29      387203.646     1871620.846      388089.062
      1871409.04      388924.132     1871844.804      389677.604
     1871714.595      390408.507     1872134.734      391064.834
     1872036.327      391902.295     1872494.109      393031.771
     1872603.484      394498.785     1872959.387       395108.16
     1872882.412      396068.058     1873389.943      396974.479
     1873212.561      397776.835     1874391.679      399797.396
      1875511.47       400648.09     1875429.873      401675.868
     1876450.707      403503.993     1876551.401      404332.118
     1877198.817      404787.617     1877735.429      405550.868
     1877737.165      406318.229      1879526.18      409377.162
     1880072.815      409612.303     1881504.526      410906.771
     1881536.059      413721.111     1882950.965      415075.671

Type RM Length L Ch R = 1 ,40107.8 ,293.6,299.9,304.4
XS GIS Cut Line= 3
     1873504.318      380855.319     1873875.891      381027.436
     1874247.463      381199.552
#Sta/Elev= 30
       0 1514.05      40 1505.54    49.9 1502.28    59.9 1496.83    69.9 1489.52
    99.9 1466.43   149.8 1426.96   169.8 1412.01   179.8 1405.34   199.8 1393.42
   219.7 1382.72   239.7  1372.8   319.6 1336.58   339.6 1326.36   359.6 1315.36
   379.5 1305.61   389.5 1301.71     402 1300.08   409.5 1299.99     417 1300.21
   499.4 1305.46   529.4 1309.59   549.3 1314.71   599.3 1330.87   629.2 1337.81
   639.2 1340.65   699.2 1361.71   729.1 1371.19     779  1383.1     819 1391.89
#Mann= 3 , 0 , 0
       0      .1       0     402    .045       0     417      .1       0
Bank Sta=402,417
XS Rating Curve= 0 ,0
Exp/Cntr=0.3,0.1

Type RM Length L Ch R = 1 ,39807.8 ,295.3,299.9,306.4
XS GIS Cut Line= 3
     1873426.217      381018.613     1873745.176      381296.666
     1874073.859      381536.859
#Sta/Elev= 30
       0 1496.67    19.7 1488.53    39.4 1478.63    68.9 1460.81   108.2  1434.1
   167.3 1392.71   255.8 1328.55   275.5 1313.32   285.4 1307.12   295.2 1303.61
   305.1 1301.82   354.3 1297.13   415.6 1288.35   423.1 1287.62   430.6 1288.26
   492.6 1302.73   522.4 1310.49   542.3 1316.71   562.2 1324.83   572.1 1329.98
     582 1335.75   611.8 1355.31   631.6 1366.41   711.1 1401.72   730.9 1409.05
   770.7 1417.09   780.6 1420.09   790.5 1426.08   800.4 1434.64   830.2 1465.35
#Mann= 3 , 0 , 0
       0      .1       0   415.6    .045       0   430.6      .1       0
Bank Sta=415.6,430.6
XS Rating Curve= 0 ,0
Exp/Cntr=0.3,0.1

Type RM Length L Ch R = 1 ,39507.8 ,299.9,300,300.2
XS GIS Cut Line= 3
     1873252.779      381144.889      1873501.93      381469.872
     1873751.082      381794.855
#Sta/Elev= 30
       0 1499.75      20 1486.35      40 1470.52    69.9 1445.52   119.8 1401.87
   139.8 1385.69   159.8 1370.61   189.8 1349.18   209.7 1335.95   229.7 1323.86
   249.7 1312.78   269.7 1302.92   279.7 1300.17   369.6 1290.04   389.5 1283.26
   399.5 1281.09     402 1281.11     417 1282.07   469.4 1290.19   549.3 1310.52
   569.3 1316.23   589.3 1325.13   659.2 1362.24   729.1 1398.38   739.1 1402.46
   749.1  1405.2     789 1412.56     799 1417.45     809 1426.07     819 1435.62
#Mann= 3 , 0 , 0
       0      .1       0     402    .045       0     417      .1       0
Bank Sta=402,417
XS Rating Curve= 0 ,0
Exp/Cntr=0.3,0.1

Type RM Length L Ch R = 1 ,39207.8 ,164.4,159,153.5
XS GIS Cut Line= 3
      1873028.88       381341.68     1873277.527      381667.732
     1873523.169      381995.255
#Sta/Elev= 30
       0 1440.97      40  1412.4     160 1332.67     210 1301.31     220 1297.11
     230 1294.68     250 1291.82   402.5 1273.91     410 1273.66   417.5 1273.99
     430 1275.82     450 1281.79     460 1283.85   519.9 1287.16   529.9 1288.46
   539.8 1290.94   549.8 1294.76   559.8 1300.32   569.8 1307.36   579.8 1315.71
   589.8 1324.96   629.7 1364.57   649.7 1381.62   659.7 1388.31   669.7 1394.06
   689.6  1402.4   699.6 1405.26   749.6  1415.9   759.5 1420.45   819.4 1463.56
#Mann= 3 , 0 , 0
       0      .1       0   402.5    .045       0   417.5      .1       0
Bank Sta=402.5,417.5
XS Rating Curve= 0 ,0
Exp/Cntr=0.3,0.1

Type RM Length L Ch R = 1 ,39048.6 ,137.6,128,118.4
XS GIS Cut Line= 3
      1872887.69      381505.047     1873055.251      381679.663
     1873475.116       382031.65
#Sta/Elev= 30
       0 1373.45    19.4  1364.1    58.1 1344.33   116.2 1322.61   183.9 1295.07
   203.3 1288.42   232.3  1281.5     252 1278.84   281.8 1278.04   321.7 1274.31
   350.2 1273.66   365.2 1273.66   381.5 1273.86   391.4 1274.81   481.1 1289.43
     491 1291.92     501 1297.69     511 1304.94   560.8 1343.58   620.6 1391.16
   630.5 1398.42   640.5 1402.78   650.4 1404.82   660.4 1405.82   720.2 1405.58
     750 1407.07     760 1408.14     770 1410.89   779.9 1416.73   789.9 1424.45
#Mann= 3 , 0 , 0
       0      .1       0   350.2    .045       0   365.2      .1       0
Bank Sta=350.2,365.2
XS Rating Curve= 0 ,0
Exp/Cntr=0.3,0.1

Type RM Length L Ch R = 1 ,38920.6 ,102.4,104.7,107
XS GIS Cut Line= 4
     1872719.455      381689.252     1872923.123      381816.545
     1873184.652      381885.977     1873323.516      381973.925
#Sta/Elev= 30
       0 1400.66      50 1371.96    80.1 1356.02   110.1 1340.89   180.1 1306.41
   220.2  1287.2   230.2 1282.71   240.2 1279.09   249.8 1276.65   259.5 1275.03
   269.2 1274.28   327.2 1273.66   389.3 1273.66   404.3 1273.66   414.1 1273.67
   423.8 1274.05   433.4 1275.21   462.4 1279.48   491.4  1284.9   501.1 1287.08
   510.8 1290.31   520.4  1295.7   530.1 1302.58   578.4 1337.96   607.4 1358.49
   617.1 1365.03   626.8 1371.46   646.1 1383.74   665.5    1395   675.1 1399.56
#Mann= 3 , 0 , 0
       0      .1       0   389.3    .045       0   404.3      .1       0
Bank Sta=389.3,404.3
XS Rating Curve= 0 ,0
Exp/Cntr=0.3,0.1

Type RM Length L Ch R = 1 ,38815.8 ,70.4,68.6,66.7
XS GIS Cut Line= 4
      1872664.26      381776.569      1872870.91      381888.673
     1873119.429      381983.219     1873280.157       382048.05
#Sta/Elev= 30
       0  1400.1    58.8 1362.73    78.4 1351.02   156.7  1311.2   205.7 1284.52
   215.5 1280.26   225.3 1277.16   235.1 1274.94     245 1274.15   343.4 1274.12
   363.1 1275.49   382.8 1278.28   392.7 1278.18   402.5 1274.87   422.2 1261.58
   426.1 1260.34   432.1 1258.42   441.1 1257.48   451.8 1257.12   461.6 1258.34
   471.4 1263.03     501 1283.92   510.6 1291.58   539.5 1315.95   549.1 1323.12
   558.8 1329.47     578 1340.34   635.8 1370.85     655 1380.61   674.3 1389.26
#Mann= 3 , 0 , 0
       0      .1       0   426.1    .045       0   441.1      .1       0
Bank Sta=426.1,441.1
XS Rating Curve= 0 ,0
Exp/Cntr=0.3,0.1

Type RM Length L Ch R = 1 ,38747.3 ,289,289.5,290
XS GIS Cut Line= 3
      1872686.16      381898.967     1872786.108      381951.642
     1873234.524      382082.655
#Sta/Elev= 30
       0 1349.38     9.4 1340.95    28.2 1325.66    47.1 1312.65    84.7 1292.19
   103.6 1282.61     113 1278.83   122.9 1275.95   132.9 1274.43   142.8 1274.07
     282 1274.09   291.9 1274.46   301.8 1275.74   321.7 1279.29   331.6 1278.46
   341.6 1274.83   351.5 1269.06   361.5 1262.37     366 1260.45   371.4 1258.14
     381 1258.89   421.1 1273.93     441 1284.64   460.9  1297.1   470.8 1303.95
   520.5 1341.03   540.4 1354.78   550.3 1360.96   560.3 1366.58   580.1 1376.64
#Mann= 3 , 0 , 0
       0      .1       0     366    .045       0     381      .1       0
Bank Sta=366,381
XS Rating Curve= 0 ,0
Exp/Cntr=0.3,0.1

Type RM Length L Ch R = 1 ,38457.8 ,148.6,150,150.9
XS GIS Cut Line= 3
     1872563.606      382178.968     1872954.098      382302.282
      1873344.59      382425.595
#Sta/Elev= 30
       0 1290.75    69.9 1286.56   109.9  1290.1   129.8 1289.77   189.8 1277.32
   209.7 1274.48   309.6 1274.18   319.6 1274.88   339.6 1278.07   349.6 1277.71
   359.6 1274.37   389.5  1259.8   399.5 1255.45     402 1255.06   409.5  1253.9
     417 1255.31   429.5 1260.18   509.4 1298.01   549.3 1318.47   569.3 1330.67
   579.3 1337.96   619.2 1370.59   649.2 1392.79   659.2 1398.27   719.1 1422.49
   729.1 1427.74   739.1 1435.25     779 1471.25     809  1497.4     819 1505.36
#Mann= 3 , 0 , 0
       0      .1       0     402    .045       0     417      .1       0
Bank Sta=402,417
XS Rating Curve= 0 ,0
Exp/Cntr=0.3,0.1

Type RM Length L Ch R = 1 ,38307.8 ,301.4,300,299.5
XS GIS Cut Line= 3
     1872524.882      382297.613     1872909.965      382445.515
     1873294.854      382583.776
#Sta/Elev= 30
       0 1291.65    78.6  1287.3     108 1290.23   117.9 1290.16   147.3 1283.65
   196.4 1277.44   294.6 1268.37   343.8 1265.47   363.4 1261.55   392.9 1252.56
   402.7 1250.43     405 1250.46   412.5 1250.57     420  1252.6   432.5 1257.67
   452.4 1267.28   512.3 1302.19   572.1 1338.78     612 1364.81   641.9 1385.58
   651.9 1391.18   661.9 1393.89   691.8 1396.03   701.8 1398.05   711.8  1401.2
   721.7 1405.75   731.7  1412.4   741.7 1420.83   771.6 1449.45   821.5 1488.88
#Mann= 3 , 0 , 0
       0      .1       0     405    .045       0     420      .1       0
Bank Sta=405,420
XS Rating Curve= 0 ,0
Exp/Cntr=0.3,0.1

Type RM Length L Ch R = 1 ,38007.8 ,298.8,300,300.8
XS GIS Cut Line= 3
      1872398.89      382593.615     1872789.671      382716.265
     1873178.144      382845.756
#Sta/Elev= 30
       0 1383.62      10 1378.72    69.9 1345.26   169.8 1293.24   199.8 1278.92
   229.8 1266.69   269.7 1253.75   299.7 1248.29   319.7 1246.43   349.6 1248.68
   359.6 1248.17   402.1 1240.36   409.6 1239.84   417.1 1240.96   419.6 1241.34
   429.6 1245.74   439.5 1251.45   469.5 1266.63   499.5 1284.31   589.4  1339.6
   599.3 1346.57   609.3 1354.78   639.3 1385.64   649.3 1391.58   709.2 1402.05
   719.2 1406.23   729.2 1413.25   739.2 1422.02   779.1 1459.72   819.1 1495.11
#Mann= 3 , 0 , 0
       0      .1       0   402.1    .045       0   417.1      .1       0
#XS Ineff= 2 , 0
          344.55 1252.68
Permanent Ineff=
       F       F
Bank Sta=402.1,417.1
XS Rating Curve= 0 ,0
Exp/Cntr=0.3,0.1

Type RM Length L Ch R = 1 ,37707.8 ,453.3,450,446.9
XS GIS Cut Line= 3
      1872306.69      382855.462     1872690.117      382999.247
     1873073.543      383143.032
#Sta/Elev= 30
       0 1361.37    69.9  1334.9   119.8 1318.38   169.8 1303.82   239.7 1287.87
   269.7 1279.77   309.6  1266.1   329.6  1257.6   349.6 1248.04   359.6 1244.49
     402 1236.77   409.5 1236.41     417 1237.63   429.5 1242.06   459.4 1255.35
   479.4 1266.59   529.4 1297.99   649.2  1377.7   659.2 1384.12   669.2 1389.54
   679.2 1392.57   709.1 1394.39   719.1 1395.71   729.1 1400.91   739.1 1411.46
     779 1462.44     789 1474.92     799 1486.28     809 1495.43     819 1502.07
#Mann= 3 , 0 , 0
       0      .1       0     402    .045       0     417      .1       0
Bank Sta=402,417
XS Rating Curve= 0 ,0
Exp/Cntr=0.3,0.1

Type RM Length L Ch R = 1 ,37257.8 ,304.7,300,294.9
XS GIS Cut Line= 3
     1872159.508      383342.531     1872560.256      383428.357
     1872959.423      383518.903
#Sta/Elev= 30
       0 1359.94      80 1316.64   189.9 1258.81   209.9 1248.88   219.9 1245.44
   229.9 1244.02   289.9 1244.59   299.9 1244.02   309.9 1242.42   349.9  1233.7
   389.8 1222.95   402.3 1220.43   409.8 1219.84   417.3 1220.38   429.8 1222.32
   459.8 1228.86   479.7 1236.15   509.7 1249.23   529.6 1258.69   559.6 1273.76
   599.5  1294.9   629.5 1311.93   649.4 1324.88   679.4 1348.05   719.3 1382.04
   729.3 1389.79   739.3 1395.42   749.3 1398.45   759.2    1400   819.1    1407
#Mann= 3 , 0 , 0
       0      .1       0   402.3    .045       0   417.3      .1       0
Bank Sta=402.3,417.3
XS Rating Curve= 0 ,0
Exp/Cntr=0.3,0.1

Type RM Length L Ch R = 1 ,36957.8 ,279.2,283.4,287.3
XS GIS Cut Line= 3
     1872095.026      383721.579     1872504.526      383721.579
     1872914.026      383721.579
#Sta/Elev= 30
       0 1396.02      10 1390.67      40 1376.25    79.9 1353.68   109.9  1335.8
   129.8 1325.02   169.8 1305.42   249.7 1268.18   289.6 1250.44   309.6 1243.05
   359.6  1225.7   369.6  1221.6   379.5 1216.54   389.5 1212.27   399.5 1210.69
     402 1210.87   409.5 1211.41     417 1212.84   449.4    1219   509.4 1229.23
   519.4 1231.69   529.4 1235.67   609.3 1276.64   639.2 1292.67   669.2 1309.28
   739.1 1350.26   759.1 1361.28     799 1381.42     809 1386.08     819 1389.96
#Mann= 3 , 0 , 0
       0      .1       0     402    .045       0     417      .1       0
Bank Sta=402,417
XS Rating Curve= 0 ,0
Exp/Cntr=0.3,0.1

Type RM Length L Ch R = 1 ,36674.3 ,318.3,320.6,323.2
XS GIS Cut Line= 3
     1872056.791      383922.925     1872454.262      383998.689
     1872864.473      384070.219
#Sta/Elev= 30
       0  1305.9      79 1290.83    88.8 1288.32   108.6 1280.94   118.4 1278.98
   128.3 1278.86   167.8  1281.5   187.5 1282.16   207.2 1281.87   217.1 1281.07
     227 1279.24   246.7 1272.33   355.3 1223.71     375 1215.86   394.8 1206.94
     402 1205.22   404.6  1204.6     417    1205   454.2  1207.1   464.1 1208.19
     474 1210.18   493.9 1216.56   523.6  1228.6   543.4 1235.32   573.2 1241.14
   672.3 1277.19   692.1 1286.17   731.8 1306.06   761.5 1319.22     821 1336.95
#Mann= 3 , 0 , 0
       0      .1       0     402    .045       0     417      .1       0
Bank Sta=402,417
XS Rating Curve= 0 ,0
Exp/Cntr=0.3,0.1

Type RM Length L Ch R = 1 ,36353.6 ,175.5,178.3,181
XS GIS Cut Line= 3
     1872008.369      384192.736     1872446.741      384323.591
     1872607.247       384434.71
#Sta/Elev= 30
       0 1332.02    79.6 1290.05   129.3 1263.15   139.2 1258.34   149.2  1254.7
   198.9 1240.21   248.6 1224.14   268.5 1218.86   278.5 1216.62   288.4 1214.63
   308.3 1211.22   318.2 1209.97   348.1 1207.47   377.9 1203.77   387.9 1202.12
   407.8 1197.22   410.9 1196.76   417.7 1195.76   425.9  1196.2   427.6 1196.29
   437.6 1199.32   467.2 1214.86     516 1241.96   525.8 1247.89   545.3 1260.62
   564.8 1271.58   584.4 1281.68   613.7 1295.68   633.2 1305.99   652.7 1316.71
#Mann= 3 , 0 , 0
       0      .1       0   410.9    .045       0   425.9      .1       0
Bank Sta=410.9,425.9
XS Rating Curve= 0 ,0
Exp/Cntr=0.3,0.1

Type RM Length L Ch R = 1 ,36175.3 ,142.6,147.9,154
XS GIS Cut Line= 4
     1871981.099      384339.466     1872280.945      384450.585
     1872361.343        384485.6     1872700.728      384605.799
#Sta/Elev= 30
       0 1328.19      40 1307.23      70 1291.09    99.9 1274.05   189.9    1224
   199.9 1218.49   209.8 1213.79   219.8 1210.84   229.8 1209.28   279.8 1203.18
   319.8 1200.44   329.5 1199.49   339.3 1197.73     349 1195.34   358.8 1194.15
   364.2 1194.21   379.2 1194.25     388 1194.39   397.7 1196.25   407.5 1199.98
   427.5 1208.96   447.5 1218.52   457.5 1223.59   477.5 1234.41   497.5 1245.93
   547.5 1275.75   587.5 1298.96   607.5 1311.04   727.5 1385.67   767.5 1411.95
#Mann= 3 , 0 , 0
       0      .1       0   364.2    .045       0   379.2      .1       0
Bank Sta=364.2,379.2
XS Rating Curve= 0 ,0
Exp/Cntr=0.3,0.1

Type RM Length L Ch R = 1 ,36027.4 ,121.9,119.6,118.6
XS GIS Cut Line= 4
     1871949.827      384396.346     1872128.821      384498.628
     1872292.079      384630.415     1872553.686      384744.499
#Sta/Elev= 30
       0 1333.87    29.4 1316.24    68.7 1293.33   117.8  1265.7   176.7 1231.91
   196.3 1221.36   206.2 1216.54   226.1 1208.18   246.1 1201.19   256.1 1198.79
   266.1 1197.96   296.1 1198.91   316.1 1198.31     336 1195.45     346 1194.29
   349.9 1194.28     356 1194.26   364.9 1194.26     386 1194.52     396 1195.57
     416 1199.72   425.8 1202.26   435.6 1205.44   445.5 1209.62   534.1 1256.38
   563.6 1272.62     603 1295.08   632.5 1312.55   652.2 1324.85   701.4 1358.28
#Mann= 3 , 0 , 0
       0      .1       0   349.9    .045       0   364.9      .1       0
#XS Ineff= 2 , 0
          289.11 1205.34
Permanent Ineff=
       F       F
Bank Sta=349.9,364.9
XS Rating Curve= 0 ,0
Exp/Cntr=0.3,0.1

Type RM Length L Ch R = 1 ,35907.8 ,308.7,300,289.3
XS GIS Cut Line= 3
     1871806.633      384452.587     1872153.751      384663.338
     1872499.118      384917.549
#Sta/Elev= 30
       0 1388.25    19.8 1374.88    39.6 1362.41    69.3 1344.87    89.1 1333.87
   118.8 1318.12   148.6 1303.13   198.1 1279.18   227.8 1265.44   336.8  1203.8
   346.7 1199.56   366.5 1195.89   376.4 1192.88   396.2 1184.86   398.6 1184.53
   406.1 1183.48   413.6 1183.61     426 1185.34     446 1191.51   505.8 1198.83
   535.7 1203.61   545.7 1205.93   555.7 1210.35   635.5 1257.84   655.4 1269.05
   675.4 1279.58   725.2 1302.84     805 1335.99     815  1341.1   834.9 1352.27
#Mann= 3 , 0 , 0
       0      .1       0   398.6    .045       0   413.6      .1       0
Bank Sta=398.6,413.6
XS Rating Curve= 0 ,0
Exp/Cntr=0.3,0.1

Type RM Length L Ch R = 1 ,35607.8 ,149,150,151.1
XS GIS Cut Line= 3
     1871658.739      384881.719     1872063.014      384946.924
     1872467.289      385012.128
#Sta/Elev= 30
       0 1427.83      20 1414.22      40 1398.84    59.9 1381.87   109.9 1337.37
   139.8 1312.36   159.8 1297.33   209.7 1261.58   219.7 1255.46   229.7 1250.49
   259.7 1237.26   349.6 1199.88   379.5 1188.07   389.5 1183.58   399.5 1180.13
     402 1179.84     417 1178.83   449.4 1177.02   479.4  1178.4   499.4 1180.55
   519.4 1184.57   529.4 1188.39   559.3  1205.1   639.2 1253.51   679.2 1275.94
   699.2 1286.07   749.1  1308.4   769.1 1317.87     799 1333.88     819 1345.81
#Mann= 3 , 0 , 0
       0      .1       0     402    .045       0     417      .1       0
Bank Sta=402,417
XS Rating Curve= 0 ,0
Exp/Cntr=0.3,0.1

Type RM Length L Ch R = 1 ,35457.8 ,154.4,149.9,145.1
XS GIS Cut Line= 3
     1871637.581      385012.151     1872038.638      385094.917
     1872439.224      385179.888
#Sta/Elev= 30
       0 1353.67      10 1350.14      30 1346.13    59.9 1342.61    79.9 1344.18
    89.9 1342.86    99.9 1338.62   119.9  1324.1   149.8  1296.4   169.8 1279.82
   269.7  1208.1   289.6 1196.14   299.6 1192.43   309.6 1190.92   349.6 1191.77
   369.6 1190.69   379.5 1188.09     402 1178.05     417 1176.56   449.5 1174.48
   469.4  1176.3   509.4    1184   519.4 1187.03   529.4 1191.66   559.3 1209.29
   599.3 1234.64   639.2 1252.77   719.1 1291.85   759.1  1315.4     819 1354.15
#Mann= 3 , 0 , 0
       0      .1       0     402    .045       0     417      .1       0
Bank Sta=402,417
XS Rating Curve= 0 ,0
Exp/Cntr=0.3,0.1

Type RM Length L Ch R = 1 ,35307.8 ,295.2,312.2,329.5
XS GIS Cut Line= 3
     1871600.495      385238.623     1872007.998      385241.098
     1872428.816      385238.883
#Sta/Elev= 30
       0 1343.12    49.7 1325.04    79.5 1311.72   149.1 1275.74   178.9 1258.43
   218.7 1242.69   228.6 1237.15   258.4    1218   298.2 1196.45   308.1 1192.85
   318.1 1191.18   367.8  1186.7   377.7 1183.77   387.6 1179.08     400 1175.02
   407.5 1174.15     415 1174.33   436.9 1174.98   466.2 1174.02   485.8 1174.55
     525 1179.57   534.7 1181.62   544.5  1186.3   554.3 1193.25   583.7 1219.17
   603.2 1231.28   642.4 1253.06   691.3 1276.39   720.7  1291.4   828.3 1350.73
#Mann= 3 , 0 , 0
       0      .1       0     400    .045       0     415      .1       0
Bank Sta=400,415
XS Rating Curve= 0 ,0
Exp/Cntr=0.3,0.1

Type RM Length L Ch R = 1 ,34995.7 ,292.8,287.5,280.4
XS GIS Cut Line= 4
     1871592.973      385290.866      1871921.32      385478.493
     1871987.336      385541.035      1872240.98      385730.399
#Sta/Elev= 30
       0 1318.32    39.8 1295.08   119.4 1253.72   129.4 1249.53   149.3 1245.11
   179.1 1231.66   218.9 1216.98   228.9 1212.27   278.6 1183.76   288.6  1180.5
   298.6 1179.07   378.2 1176.52   405.4 1167.32   423.6 1165.63   428.9 1166.18
   443.9 1168.14   488.9 1173.95   518.6 1176.38   528.5 1179.08   538.4 1187.52
     568 1221.46   577.9 1230.38   607.6 1253.09   627.4 1270.08     667 1306.71
   686.7  1321.3   696.6 1325.23   706.5 1325.27   716.4 1323.44   785.6 1304.12
#Mann= 3 , 0 , 0
       0      .1       0   428.9    .045       0   443.9      .1       0
Bank Sta=428.9,443.9
XS Rating Curve= 0 ,0
Exp/Cntr=0.3,0.1

Type RM Length L Ch R = 1 ,34707.8 ,308.5,300,293.3
XS GIS Cut Line= 3
     1871436.488      385538.233     1871789.538      385741.916
     1872169.625      385921.352
#Sta/Elev= 30
       0 1260.27    39.8 1241.81    99.4 1208.73   109.4 1204.17   119.3  1201.6
   149.1 1199.24   159.1 1195.66   178.9 1183.79   188.9 1179.27   198.8 1176.22
   218.7 1172.58   228.6 1171.98   298.2 1172.58   377.8 1168.43   400.1 1162.53
   407.6 1161.23   415.1 1161.54   457.6 1170.56   467.6 1174.09   527.7 1215.06
   537.7 1220.73   557.7 1227.73   587.7 1230.83   607.7 1228.93   637.8 1222.93
   647.8 1222.37   657.8 1224.44   677.8 1232.51   717.8  1251.7   827.9 1309.32
#Mann= 3 , 0 , 0
       0      .1       0   400.1    .045       0   415.1      .1       0
Bank Sta=400.1,415.1
XS Rating Curve= 0 ,0
Exp/Cntr=0.3,0.1

Type RM Length L Ch R = 1 ,34407.7 ,150.8,149.6,145.6
XS GIS Cut Line= 3
     1871324.195      385967.081     1871772.972      386034.472
     1872065.762      386002.724
#Sta/Elev= 30
       0 1235.88    19.7 1228.29    78.9 1202.84    88.8 1199.34   128.2 1187.19
   177.6 1175.14   197.3 1170.94     217  1168.1   226.9 1167.57   305.8  1167.4
     365 1164.71   384.8 1162.99   394.6 1161.37   415.4  1155.9   424.2 1154.68
   430.4 1155.12   434.1 1155.38   443.9 1157.99   463.6 1164.85   473.4 1168.96
   502.9 1185.79   512.7 1189.81   522.5 1192.39   571.6 1201.11   581.4 1203.28
   591.2 1206.36   601.1 1210.58   669.8 1244.08   728.7  1273.6   748.3 1284.13
#Mann= 3 , 0 , 0
       0      .1       0   415.4    .045       0   430.4      .1       0
Bank Sta=415.4,430.4
XS Rating Curve= 0 ,0
Exp/Cntr=0.3,0.1

Type RM Length L Ch R = 1 ,34257.8 ,131.9,129.1,128.9
XS GIS Cut Line= 3
      1871293.53      386131.809     1871695.876      386171.437
     1872133.963      386157.956
#Sta/Elev= 30
       0 1301.75    19.7 1298.45    49.3 1295.91    78.9 1297.07   128.2 1301.28
     138 1300.41   147.9 1296.73   157.8 1289.99   197.2 1254.38   226.8 1231.85
   246.5 1218.58   315.6 1174.24   325.4 1168.49   335.3 1164.46   345.1 1162.25
   374.7 1159.27   396.8 1154.54   404.3 1153.59   411.8 1154.23   434.2 1157.22
   503.9 1161.37   553.7 1165.94   563.7 1167.68   623.4 1183.67   633.4  1187.6
   643.4 1193.62   663.3 1207.64   673.2 1213.55     743 1251.59   842.6 1308.93
#Mann= 3 , 0 , 0
       0      .1       0   396.8    .045       0   411.8      .1       0
Bank Sta=396.8,411.8
XS Rating Curve= 0 ,0
Exp/Cntr=0.3,0.1

Type RM Length L Ch R = 1 ,34128.7 ,166.2,170.8,178.4
XS GIS Cut Line= 3
     1871559.419      386302.244     1871735.331      386296.133
     1872157.479      386274.349
#Sta/Elev= 30
       0 1222.85    39.1 1195.93    58.7 1182.96    68.4 1176.89      88 1165.47
    97.8 1160.66   107.6 1157.63   117.4 1156.44   136.9 1155.42   158.3 1152.48
   166.2 1152.11   173.3 1152.86     176 1153.14   185.8 1154.96   195.7 1155.99
   225.2  1156.4     235 1156.89     294 1160.55   323.5 1162.82   333.3 1164.29
   343.1 1166.82     353 1170.08   362.8 1173.93   372.6 1178.38   382.5 1183.44
   392.3 1189.14   421.8  1208.5   441.4 1220.88   520.1 1267.73   598.7 1315.02
#Mann= 3 , 0 , 0
       0     .06       0   158.3    .045       0   173.3     .06       0
Bank Sta=158.3,173.3
XS Rating Curve= 0 ,0
Exp/Cntr=0.3,0.1

Type RM Length L Ch R = 1 ,33957.8 ,232.4,246.9,258.7
XS GIS Cut Line= 3
     1871314.164      386369.067     1871781.543      386451.751
     1872162.176      386567.215
#Sta/Elev= 30
       0 1309.91   118.7 1249.79   138.4 1240.63   168.1 1227.86   247.2 1186.76
   276.9 1172.88   316.4 1156.37   326.3 1153.74   336.2 1152.89   435.1 1153.44
     445 1152.83   454.9 1150.18   467.1 1146.13   474.6 1144.61   482.1 1145.08
   484.6 1145.24   494.5 1148.64   504.5 1153.52   514.4 1157.39   524.4 1159.48
   554.2 1163.17   564.1 1165.37     584 1171.91   603.9 1180.77   613.8 1185.88
   643.7 1202.79   683.5 1224.01   693.4 1229.85     773 1280.72   872.4 1341.17
#Mann= 3 , 0 , 0
       0     .06       0   467.1    .045       0   482.1     .06       0
Bank Sta=467.1,482.1
XS Rating Curve= 0 ,0
Exp/Cntr=0.3,0.1

Type RM Length L Ch R = 1 ,33710.8 ,201.8,203.1,201.6
XS GIS Cut Line= 2
     1871458.404      386447.617     1871855.775      386873.245
#Sta/Elev= 30
       0 1210.68    39.5  1185.9      79 1160.66    88.8 1154.92    98.7 1150.95
   108.6 1149.84   128.3 1149.74   187.5 1147.45   246.7 1145.59   256.6 1144.66
   266.5 1142.16   276.3 1139.11   280.1  1138.5   286.2 1137.52   295.1  1138.4
     306  1140.6   315.8 1143.04   335.6  1147.2   345.4 1149.77   355.3 1154.45
   365.2 1161.62   384.9 1178.29   414.5 1203.78     454 1237.48   483.6 1262.42
   513.2 1286.96   532.9 1302.87   552.7 1318.14   572.4 1332.63   582.3 1339.51
#Mann= 3 , 0 , 0
       0     .06       0   280.1    .045       0   295.1     .06       0
Bank Sta=280.1,295.1
XS Rating Curve= 0 ,0
Exp/Cntr=0.3,0.1

Type RM Length L Ch R = 1 ,33507.8 ,269.8,255.9,244.8
XS GIS Cut Line= 3
     1871239.666      386477.262     1871509.538      386797.299
      1871807.13      387076.025
#Sta/Elev= 30
       0 1293.37    99.7 1230.28   209.3 1158.92   219.3 1152.76   229.2  1148.7
   239.2 1147.46   249.2 1147.51   259.2 1147.16   348.9 1140.33   388.7 1138.07
   398.7 1136.31   411.1 1133.12   418.6  1131.6   426.1  1131.8   428.6 1131.87
   438.5 1133.56   448.5 1135.59   468.4 1139.05   478.3 1141.14   488.2 1144.69
   498.2 1149.82   518.1 1162.23     538 1173.87   607.6 1210.28   617.5 1215.72
   627.5 1221.56   657.3 1239.86   736.9 1289.72   756.8 1302.58   826.4 1348.46
#Mann= 3 , 0 , 0
       0     .06       0   411.1    .045       0   426.1     .06       0
Bank Sta=411.1,426.1
XS Rating Curve= 0 ,0
Exp/Cntr=0.3,0.1

Type RM Length L Ch R = 1 ,33251.5 ,198.4,194,190.8
XS GIS Cut Line= 3
      1871129.91      386913.866     1871372.304      386977.539
     1871721.552      387021.597
#Sta/Elev= 30
       0 1191.94    19.3 1181.85    28.9 1177.64    86.8  1155.2     106 1146.35
   115.7 1142.48   125.3  1140.7   144.6 1140.51   154.2 1139.72   173.5 1136.38
   192.8 1133.74   202.4 1131.68   218.2 1126.68   221.7 1125.67   231.3 1126.01
   233.2 1126.49   250.6 1130.41   260.4 1130.95   309.3 1130.62   348.4 1132.25
     368 1133.64   387.5 1135.59   397.3 1137.05   407.1 1139.28   416.8 1142.94
   426.6 1148.34     456 1166.48   475.5 1179.71   534.2 1223.06   602.6 1275.19
#Mann= 3 , 0 , 0
       0     .06       0   218.2    .045       0   233.2     .06       0
Bank Sta=218.2,233.2
XS Rating Curve= 0 ,0
Exp/Cntr=0.3,0.1

Type RM Length L Ch R = 1 ,33057.8 ,153.4,150,145.3
XS GIS Cut Line= 3
      1870909.76      387135.897      1871317.93      387161.408
     1871727.542      387210.361
#Sta/Elev= 30
       0 1344.39      20 1330.13    49.9 1306.79    79.8 1282.24   139.6 1231.29
   159.6 1214.69   219.4 1166.51   229.4 1159.94   239.4 1155.62   259.3 1149.24
   289.3 1140.82   309.2 1136.72   319.2 1135.41   349.1 1134.26   359.1 1133.15
   369.1 1131.14     389 1123.95     399 1121.13   401.5    1121     409 1120.62
   416.5 1121.54   438.4 1125.13   566.1 1132.19   575.9 1133.95   585.8  1138.5
   595.6  1145.1     684 1209.25   752.7 1260.23   782.2 1280.99   821.5 1307.63
#Mann= 3 , 0 , 0
       0     .06       0   401.5    .045       0   416.5     .06       0
Bank Sta=401.5,416.5
XS Rating Curve= 0 ,0
Exp/Cntr=0.3,0.1

Type RM Length L Ch R = 1 ,32907.8 ,159.3,157.5,155.6
XS GIS Cut Line= 3
     1870914.094      387347.353     1871321.986      387311.098
     1871729.878      387274.842
#Sta/Elev= 30
       0 1283.08    49.9 1252.05    69.9 1240.28   189.8 1174.69   219.7 1159.02
   229.7 1155.19   239.7 1152.68   269.7 1148.04   279.7 1145.29   309.6 1132.18
   319.6 1129.63   329.6 1129.08   349.6 1129.69   359.6 1129.39   369.6 1127.38
   389.5 1119.14   399.5 1116.61     402 1116.56   409.5 1116.43     417 1117.39
   439.5 1120.41   509.4 1126.56   519.4 1127.76   529.4 1130.69   539.3 1136.03
   599.3  1176.1   759.1 1285.12     789 1305.97     809 1319.17     819  1325.2
#Mann= 3 , 0 , 0
       0      .1       0     402    .045       0     417      .1       0
Bank Sta=402,417
XS Rating Curve= 0 ,0
Exp/Cntr=0.3,0.1

Type RM Length L Ch R = 1 ,32750.3 ,298.1,292.6,288.1
XS GIS Cut Line= 4
     1871110.483      387491.378     1871232.387      387486.261
     1871426.614      387452.524     1871748.043      387401.307
#Sta/Elev= 30
       0 1161.27    18.8 1158.13    28.2 1155.84    37.5 1152.49    56.3 1143.22
    65.7 1139.75    75.1  1137.6   112.6 1132.12   141.7 1125.77     191 1122.68
   200.9 1120.91   220.6 1115.92   231.6 1113.72   240.3 1113.25   246.6 1114.43
   269.9 1120.51   299.4 1122.91   309.3 1124.83   319.2 1129.33     329 1136.14
   368.5 1167.82   388.2 1182.25     398 1188.18   417.8 1197.94   437.5 1208.52
   467.1 1226.22   496.7 1244.82   585.4 1297.52   624.9 1320.38   644.6 1331.09
#Mann= 3 , 0 , 0
       0      .1       0   231.6    .045       0   246.6      .1       0
Bank Sta=231.6,246.6
XS Rating Curve= 0 ,0
Exp/Cntr=0.3,0.1

Type RM Length L Ch R = 1 ,32457.8 ,220.3,219,216.7
XS GIS Cut Line= 4
     1871071.629      387851.661     1871228.071        387834.1
     1871416.973      387750.142     1871644.693      387662.086
#Sta/Elev= 30
       0 1206.82    49.2  1176.5   118.1 1132.98   127.9 1127.73   137.8 1124.04
   147.6 1121.58   167.3 1117.48   177.1 1116.31     187 1116.05   295.2 1116.14
   314.9 1115.84   324.8 1115.23   334.6 1113.54   354.3 1106.72   356.6 1106.42
   364.1 1105.44   371.6 1106.09   383.7 1108.29   403.2 1112.76     413 1115.61
   422.7 1119.52   432.5 1125.18   481.3 1161.13   510.6 1181.62   559.5 1215.25
   569.2  1221.5     579 1226.67   588.8 1229.76   598.5 1229.46   608.3 1228.31
#Mann= 3 , 0 , 0
       0      .1       0   356.6    .045       0   371.6      .1       0
Bank Sta=356.6,371.6
XS Rating Curve= 0 ,0
Exp/Cntr=0.3,0.1

Type RM Length L Ch R = 1 ,32238.6 ,222.9,233.8,244.8
XS GIS Cut Line= 4
      1871193.49       387987.65     1871510.927      387946.134
     1871560.837      387920.539      1871695.06      387846.363
#Sta/Elev= 30
       0  1155.7      10 1150.78      50  1132.1      60 1128.66      70 1127.37
     100 1125.94     120 1124.51   160.1 1121.26   200.1 1117.62   210.1 1117.06
   230.1 1116.39   240.1 1115.73   270.1 1112.96   280.1  1112.4   310.1 1111.49
   320.1 1110.79   329.5 1108.51   339.3 1105.08   348.2 1103.33   354.3 1103.96
   357.5 1104.29   366.9 1107.82   376.2 1111.68   395.4 1118.68     405  1122.7
   414.6  1127.7   424.2  1133.5   433.7 1139.58   472.1 1164.63   529.6 1203.56
#Mann= 3 , 0 , 0
       0      .1       0   339.3    .045       0   354.3      .1       0
Bank Sta=339.3,354.3
XS Rating Curve= 0 ,0
Exp/Cntr=0.3,0.1

Type RM Length L Ch R = 1 ,32004.8 ,289.8,296.9,303.9
XS GIS Cut Line= 3
      1871347.14      388158.961     1871590.861        388141.3
     1871905.225      388144.833
#Sta/Elev= 30
       0 1130.28    19.6 1128.42    97.7 1119.62   117.3 1117.23   127.1 1115.58
   156.4 1109.42   166.2 1108.11   175.9 1107.47   224.8 1105.28   234.6 1104.55
   244.4  1102.4   254.2 1099.14   258.4 1098.24     264 1097.04   273.4 1096.94
   293.5 1099.17   303.3  1100.7   313.1  1103.9     323 1109.28   332.8 1115.21
   342.6 1120.31   352.4 1124.95   362.2 1129.86   401.6 1151.24   421.2 1162.37
   470.3 1191.23   480.2 1196.66     490 1201.76   529.3 1221.33   558.7 1237.07
#Mann= 3 , 0 , 0
       0      .1       0   258.4    .045       0   273.4      .1       0
Bank Sta=258.4,273.4
XS Rating Curve= 0 ,0
Exp/Cntr=0.3,0.1

Type RM Length L Ch R = 1 ,31707.9 ,262.6,262.4,262.1
XS GIS Cut Line= 4
     1871285.327      388369.126     1871486.661      388411.513
     1871622.297      388456.725      1871921.12      388494.519
#Sta/Elev= 30
       0 1197.75    78.4 1143.84   137.2 1105.16     147 1101.32   156.8 1100.44
   186.2 1101.24     196 1101.29   205.8 1100.78   215.3 1098.62   224.8 1094.56
   234.3 1091.49   241.5 1091.15   243.9 1091.04   256.5 1093.74   262.9 1095.67
   272.5 1097.66     282  1098.3   329.7 1098.35   339.2 1098.52   348.7 1099.35
   358.4 1101.64   368.2 1105.66   377.9 1110.86   387.6 1116.64   426.4 1140.77
   533.3 1204.22   562.5 1222.02   591.6 1240.41   620.8 1259.43   649.9  1280.8
#Mann= 3 , 0 , 0
       0      .1       0   241.5    .045       0   256.5      .1       0
Bank Sta=241.5,256.5
XS Rating Curve= 0 ,0
Exp/Cntr=0.3,0.1

Type RM Length L Ch R = 1 ,31445.5 ,187.9,187.3,186.8
XS GIS Cut Line= 3
     1871144.039      388572.227     1871518.451      388692.322
     1871755.107      388759.433
#Sta/Elev= 30
       0 1216.21    19.7 1204.51   127.8 1138.66   186.8 1104.12   196.6 1098.95
   206.4  1095.7   216.3 1094.34   235.9 1093.84   265.4 1095.25   285.1 1095.22
   304.7 1093.96   334.2 1091.16   353.1 1087.98   363.7 1086.81   368.1 1086.82
   373.5 1086.84   383.4 1088.26   393.2 1091.63   412.9 1101.55   432.6 1113.23
   452.2 1126.04   481.8 1147.03     531 1183.23   540.8 1190.04   550.6 1196.25
   570.3 1207.03   599.8 1222.02   609.7 1226.73   619.5  1230.7   639.2 1237.36
#Mann= 3 , 0 , 0
       0     .06       0   353.1    .045       0   368.1     .06       0
Bank Sta=353.1,368.1
XS Rating Curve= 0 ,0
Exp/Cntr=0.3,0.1

Type RM Length L Ch R = 1 ,31257.9 ,312.7,292.9,273.1
XS GIS Cut Line= 3
     1871027.064      388737.294     1871438.977      388858.334
     1871566.135      388879.527
#Sta/Elev= 30
       0 1238.82      20 1225.82    39.9 1213.05    49.9    1207   209.7 1113.28
   229.6 1101.44   239.6 1096.04   249.6 1092.38   259.6 1090.88   309.5 1087.36
   319.5 1086.92   359.4 1086.06   369.4 1085.65   379.4  1084.2   390.2 1081.95
   399.4 1080.82   405.2 1081.44   409.4 1081.89   419.3 1085.36   429.3 1090.01
   459.1 1104.81     469 1109.89   478.9 1115.15   488.8 1120.63   508.7 1132.19
   518.6 1137.46   528.5 1142.35   538.4 1146.79   548.3 1150.85   558.2 1154.73
#Mann= 3 , 0 , 0
       0     .06       0   390.2    .045       0   405.2     .06       0
Bank Sta=390.2,405.2
XS Rating Curve= 0 ,0
Exp/Cntr=0.3,0.1

Type RM Length L Ch R = 1 ,30964.6 ,320.8,326,331.6
XS GIS Cut Line= 2
     1871272.964      389266.302     1871831.049      388893.656
#Sta/Elev= 30
       0 1168.21      10 1161.87      30  1147.1    50.1 1131.78    90.1 1100.64
   100.2 1093.09   110.2 1087.41   120.2 1085.31   190.3 1081.78   200.3 1081.67
   210.3 1081.94   280.4 1085.07   290.5 1085.12   300.5 1084.11   331.1 1078.61
   340.5 1078.16   346.1 1079.52   350.6 1080.62   370.6 1095.63   380.6 1101.35
   400.6 1111.47   420.7    1122   440.7 1133.01   530.8 1186.15   550.9 1198.53
   560.9 1205.13   580.9  1219.1     601 1234.18     621 1250.01   671.1 1290.34
#Mann= 3 , 0 , 0
       0      .1       0   331.1    .045       0   346.1      .1       0
#XS Ineff= 2 , 0
          278.39 1094.57
Permanent Ineff=
       F       F
Bank Sta=331.1,346.1
XS Rating Curve= 0 ,0
Exp/Cntr=0.3,0.1

Type RM Length L Ch R = 1 ,30638.9 ,293.9,298.9,303.7
XS GIS Cut Line= 3
     1871384.228      389469.403     1871748.043      389335.179
     1872113.624      389208.021
#Sta/Elev= 30
       0 1192.16     9.9 1187.73    19.9 1181.89    39.8 1167.62    59.7 1152.19
    79.6 1135.77   129.3 1092.98   139.2 1085.26   149.2 1080.76   159.1 1079.74
   218.8  1077.6   298.3 1070.64     348 1070.44   377.8 1069.15   380.2 1069.24
   387.8 1069.53   395.2 1071.38   407.6 1076.66   427.5 1086.67   457.3 1104.06
     487 1124.46   526.7 1154.83   546.6 1169.38   566.4  1181.7   586.3 1190.56
   635.9 1208.31   665.7 1222.38   715.3 1250.89   735.2 1263.28   774.8 1289.43
#Mann= 3 , 0 , 0
       0     .06       0   380.2    .045       0   395.2     .06       0
Bank Sta=380.2,395.2
XS Rating Curve= 0 ,0
Exp/Cntr=0.3,0.1

Type RM Length L Ch R = 1 ,30340   ,276.8,280.7,284.5
XS GIS Cut Line= 3
     1871425.896      389673.235     1871836.348      389619.521
     1872216.058      389571.836
#Sta/Elev= 30
       0 1183.42    98.6  1123.2     138 1098.26   147.8 1091.82   167.6  1077.8
   177.4    1073   187.3 1071.92   197.1 1072.36     207 1071.96   226.7 1070.11
   236.5 1069.73   374.5  1067.6   384.4 1066.68   404.1 1062.08   406.2 1061.91
     414 1061.26   421.2 1062.28   423.8 1062.65   433.6 1065.82   443.4 1069.86
   453.2 1076.73   472.8 1095.79   482.6 1104.21   492.4 1112.21   531.7 1141.71
     571 1171.76   688.7 1263.84   767.2 1323.73   786.8 1339.12   796.6 1346.53
#Mann= 3 , 0 , 0
       0      .1       0   406.2    .045       0   421.2      .1       0
Bank Sta=406.2,421.2
XS Rating Curve= 0 ,0
Exp/Cntr=0.3,0.1

Type RM Length L Ch R = 1 ,30059.3 ,300.5,307.2,313.9
XS GIS Cut Line= 3
     1871414.251       389827.92     1871790.429      389896.797
     1871993.485      389905.219
#Sta/Elev= 30
       0 1173.21      49 1138.81   127.5 1080.34   137.3  1073.5   147.1 1068.77
   156.9 1067.03   205.9 1066.79   235.3 1065.72   274.6 1058.46   294.2 1056.87
   313.8 1057.36   343.2 1060.54     353  1061.1   372.6 1061.66   382.4 1061.27
   392.1  1059.1   401.8 1055.67   406.8  1054.4   411.5 1053.21   421.8 1053.46
   430.8    1056   440.5 1060.63   450.2 1065.84   459.8 1071.85   479.2 1086.82
   498.6  1102.7     547  1145.4   566.3 1161.78     576 1169.38   585.7 1176.07
#Mann= 3 , 0 , 0
       0      .1       0   406.8    .045       0   421.8      .1       0
#XS Ineff= 2 , 0
          361.91 1067.21
Permanent Ineff=
       F       F
Bank Sta=406.8,421.8
XS Rating Curve= 0 ,0
Exp/Cntr=0.3,0.1

Type RM Length L Ch R = 1 ,29752.1 ,273.4,260.5,247.5
XS GIS Cut Line= 3
     1871398.356      390165.243     1871709.189      390177.606
     1871938.781      390258.846
#Sta/Elev= 30
       0 1130.73    48.6 1110.18    77.8  1097.4   116.6 1079.88   145.8 1067.14
   155.5 1062.49   165.3 1057.22     175 1053.55   184.7 1054.49   194.4 1057.28
   204.2 1058.56   213.9  1058.4   291.6 1054.07   301.4  1053.1   311.1 1051.28
   320.8 1048.68   327.5  1047.6   330.6  1047.1   340.3 1047.08   342.5  1047.3
     350 1048.04   359.8 1049.93   398.8 1058.18   408.5 1060.96   418.2 1065.03
     428 1070.47   457.2 1088.13   476.7 1099.06   505.9 1113.17   554.6 1135.64
#Mann= 3 , 0 , 0
       0      .1       0   327.5    .045       0   342.5      .1       0
Bank Sta=327.5,342.5
XS Rating Curve= 0 ,0
Exp/Cntr=0.3,0.1

Type RM Length L Ch R = 1 ,29491.6 ,341.8,336.4,331.1
XS GIS Cut Line= 4
     1871325.947      390488.438     1871656.206      390454.883
     1871854.009      390407.198     1871970.571      390357.748
#Sta/Elev= 30
       0 1181.18    19.5 1165.83    48.8 1143.62    68.3 1129.45    97.6 1109.19
   126.9 1090.56   146.4 1078.68   156.2 1073.18     166 1069.13   175.7 1066.75
   185.5 1065.19   224.6 1059.85   244.1 1058.04   283.1 1055.09   351.3 1048.08
   380.4 1045.72     400 1041.78   409.5 1041.48     415 1042.32   428.8 1044.72
   438.5 1045.68   496.7 1048.42   535.4 1049.59   545.2  1051.3   554.9 1055.55
   564.6  1061.4   574.4 1068.03   623.1 1102.85   642.6 1117.35     662 1132.25
#Mann= 3 , 0 , 0
       0      .1       0     400    .045       0     415      .1       0
Bank Sta=400,415
XS Rating Curve= 0 ,0
Exp/Cntr=0.3,0.1

Type RM Length L Ch R = 1 ,29155.2 ,239.9,243.2,246.4
XS GIS Cut Line= 3
     1871612.054      390868.148     1871806.324      390772.779
      1872228.42      390546.719
#Sta/Elev= 30
       0 1142.21    29.5 1125.67    78.7 1103.34    88.5 1099.58   127.9 1086.48
   147.6 1078.89   157.4 1073.33   177.1 1060.41   186.9 1055.01   196.7 1050.54
   216.4 1042.86   226.4 1039.95   236.4 1038.68   296.2 1037.05   318.7 1032.56
   326.2 1031.82   333.7 1032.05     366 1036.82   435.9 1041.17   525.6 1048.25
   535.6 1049.35   545.6  1051.8   555.6 1056.23   575.5 1066.95   585.5 1073.38
   595.5 1080.76   605.5    1089   615.4 1097.88   655.3 1136.81   695.2  1174.5
#Mann= 3 , 0 , 0
       0     .06       0   318.7    .045       0   333.7     .06       0
Bank Sta=318.7,333.7
XS Rating Curve= 0 ,0
Exp/Cntr=0.3,0.1

Type RM Length L Ch R = 1 ,28912   ,347,356.8,366.6
XS GIS Cut Line= 2
     1871744.511      391002.372     1872403.264      390779.844
#Sta/Elev= 30
       0 1121.01    59.6 1082.36   109.3 1048.34   119.2 1041.95   129.1 1037.51
   139.1 1035.82   168.9 1033.65   228.5  1032.3   268.2 1031.67     298 1031.48
   307.9 1031.12   317.9 1030.04   327.8 1028.21   337.7 1026.79   340.5 1026.73
   347.7 1026.56   355.5 1027.27   367.5 1029.08   387.4 1032.58   437.1 1040.38
     447 1043.15   456.9 1047.94   466.9 1054.13   516.5 1086.33   536.4 1100.32
   556.3 1114.85   615.9 1156.76   625.8 1163.97   635.7 1171.52   695.3 1218.06
#Mann= 3 , 0 , 0
       0     .06       0   340.5    .045       0   355.5     .06       0
Bank Sta=340.5,355.5
XS Rating Curve= 0 ,0
Exp/Cntr=0.3,0.1

Type RM Length L Ch R = 1 ,28555.2 ,292.3,292.6,292.8
XS GIS Cut Line= 3
     1871707.863      391191.584     1872168.373      391240.794
     1872523.358      391235.496
#Sta/Elev= 30
       0 1140.93    39.4  1113.2     138 1040.18   147.8 1034.88   157.7 1032.92
   177.4  1031.8   285.8 1029.01   364.6 1025.04   384.3 1023.27   404.9 1020.55
   413.9 1020.22   419.9 1020.53   433.6 1021.63   443.4 1023.03   453.3 1025.68
   463.1 1029.96     473 1035.47   482.9  1041.8   492.7 1049.02   502.6 1057.14
   532.2  1083.7     542 1091.54   561.8 1105.57   611.1 1139.05   630.8 1153.19
   640.6 1161.17   719.5 1236.57   749.1 1263.96   798.4 1308.21   818.2 1324.86
#Mann= 3 , 0 , 0
       0      .1       0   404.9    .045       0   419.9      .1       0
Bank Sta=404.9,419.9
XS Rating Curve= 0 ,0
Exp/Cntr=0.3,0.1

Type RM Length L Ch R = 1 ,28262.6 ,264.5,262.9,261.3
XS GIS Cut Line= 3
     1871714.487      391480.983     1872113.624      391528.667
     1872387.369      391484.515
#Sta/Elev= 30
       0 1131.29    19.6 1119.53    39.2 1109.16    78.4 1091.45   117.6  1072.4
   127.5    1066   147.1 1048.81   156.9 1042.95   166.7 1039.52   245.1 1023.57
   254.9  1022.2   264.7 1021.83   274.5 1022.53   294.1 1025.42   303.9 1025.78
   333.4 1022.03   343.2 1019.55     353 1016.11   363.8 1013.65   372.6 1013.62
   378.8 1015.18   392.2 1018.86     402 1019.99   491.1 1022.27     501 1024.04
   510.9 1027.79   530.7 1038.55   619.8 1091.06   649.6  1110.8   679.3 1132.78
#Mann= 3 , 0 , 0
       0      .1       0   363.8    .045       0   378.8      .1       0
Bank Sta=363.8,378.8
XS Rating Curve= 0 ,0
Exp/Cntr=0.3,0.1

Type RM Length L Ch R = 1 ,27999.7 ,204,192.1,184.4
XS GIS Cut Line= 3
     1871636.973      391766.324     1872254.844      391795.033
     1872399.731        391839.5
#Sta/Elev= 30
       0 1170.98      20 1164.55    39.9 1156.59   119.7 1118.59   159.6 1101.35
   199.5 1085.06   209.5 1080.08   219.5 1073.05   229.5  1065.1   269.4 1032.21
   279.3 1027.14   289.3 1025.44   339.2 1022.45   369.1 1019.32   379.1 1016.56
   399.1 1007.92   402.3 1007.42     409 1006.36   417.3 1007.41     439 1012.78
   458.9 1013.11   498.8 1011.38   608.6 1017.64   618.5 1019.42     628 1023.81
   637.5 1030.26   656.4 1044.64   703.8 1075.84   741.7 1097.54   770.1 1110.16
#Mann= 3 , 0 , 0
       0      .1       0   402.3    .045       0   417.3      .1       0
Bank Sta=402.3,417.3
XS Rating Curve= 0 ,0
Exp/Cntr=0.3,0.1

Type RM Length L Ch R = 1 ,27807.8 ,303.1,306.2,305
XS GIS Cut Line= 3
     1871703.254      392162.223     1872062.738      391971.112
     1872466.953       391847.27
#Sta/Elev= 30
       0 1139.26    39.7 1129.92    49.6 1127.12    59.6 1123.34    79.4 1113.39
   188.7 1051.79   218.5 1036.55   238.3 1027.92   248.2 1025.03   258.2 1023.08
   297.9 1017.35   367.4 1010.62   399.6 1002.57   407.1 1001.93   414.6 1002.74
   436.6 1008.37   446.4 1009.38   515.3  1006.8   525.1 1007.32   554.6 1010.66
   564.4 1012.44   574.3 1016.33   613.6  1041.2   643.1 1061.41   721.7 1118.19
   731.6  1123.8   741.4 1126.86   751.2 1128.18   780.7 1129.28   829.9 1134.17
#Mann= 3 , 0 , 0
       0      .1       0   399.6    .045       0   414.6      .1       0
Bank Sta=399.6,414.6
XS Rating Curve= 0 ,0
Exp/Cntr=0.3,0.1

Type RM Length L Ch R = 1 ,27501.4 ,295.9,294.6,293.3
XS GIS Cut Line= 3
     1871802.089      392386.287     1872295.532      392208.613
     1872537.487      392058.495
#Sta/Elev= 30
       0 1119.66    29.7 1104.75    59.4 1088.78   148.4  1035.9   168.2 1025.46
   178.1 1020.87     188 1017.18   207.8 1012.31   237.5 1006.68   247.4 1005.95
   356.2 1004.26   366.1 1003.04   395.8  996.21   401.9  995.59   405.7  995.21
   416.9   995.8   514.6 1005.93   524.5 1008.58   534.3    1013   553.9 1023.69
   573.6 1035.65   583.4 1042.19     603 1057.42   632.5 1084.22   661.9 1113.57
   720.8 1174.34   750.3 1202.52   760.1 1211.08   779.7 1226.72   809.2 1247.51
#Mann= 3 , 0 , 0
       0      .1       0   401.9    .045       0   416.9      .1       0
Bank Sta=401.9,416.9
XS Rating Curve= 0 ,0
Exp/Cntr=0.3,0.1

Type RM Length L Ch R = 1 ,27206.8 ,167.1,169.6,172.1
XS GIS Cut Line= 3
     1871924.198      392679.373     1872399.731      392477.059
     1872629.324      392334.006
#Sta/Elev= 30
       0 1094.83    29.8 1081.37    59.6 1069.73    69.6  1066.8    99.4 1060.58
   139.1 1050.65   149.1 1046.53   178.9 1030.04   198.8 1019.83   218.6 1011.95
   238.5 1007.78   288.2 1001.54   308.1 1000.69   347.8 1000.78   367.7   999.5
   377.6  997.83   400.4  991.89   407.5   991.1   415.4  991.56   457.2  996.91
   506.8  999.46   536.1 1002.08   565.1 1006.54   574.8 1008.95   584.4 1012.46
   603.7 1021.04   642.4 1041.15   690.7 1069.42   758.3    1111   787.3  1126.9
#Mann= 3 , 0 , 0
       0     .06       0   400.4    .045       0   415.4     .06       0
Bank Sta=400.4,415.4
XS Rating Curve= 0 ,0
Exp/Cntr=0.3,0.1

Type RM Length L Ch R = 1 ,27037.1 ,422,429.4,435.7
XS GIS Cut Line= 3
     1872178.403      392746.412     1872325.606      392688.332
     1872764.767      392556.699
#Sta/Elev= 30
       0 1055.54     9.9 1054.04    19.8 1050.25    29.7 1044.56    39.6 1038.49
      89 1006.24    98.9 1000.42   108.8  996.78   118.7  995.71   148.4  995.72
   158.2  995.39   168.2  993.13   178.2  989.99   188.2  988.82   188.5  988.84
   198.1  989.32   203.5  989.89     228  992.39     248  994.07   357.6  1001.8
   367.6 1004.02   377.5 1008.85   407.4 1027.73   447.3 1051.06   507.1 1085.32
     527 1097.19   546.9 1109.73   556.9  1115.7   576.8 1126.53   616.7 1147.58
#Mann= 3 , 0 , 0
       0     .06       0   188.5    .045       0   203.5     .06       0
Bank Sta=188.5,203.5
XS Rating Curve= 0 ,0
Exp/Cntr=0.3,0.1

Type RM Length L Ch R = 1 ,26607.8 ,316.1,312.2,309.4
XS GIS Cut Line= 3
     1872094.197      393063.402      1872497.09      393079.295
     1872902.038      393075.036
#Sta/Elev= 30
       0 1090.95    39.3 1071.73    88.5 1045.49    98.3 1039.52   108.2 1032.23
   127.8 1015.98   147.5 1001.73   157.4  996.27   167.2  992.16     177  989.08
   186.8  986.75   196.7   985.2   206.5  984.53   216.4  984.64   285.2  989.08
   304.9     989   363.9  986.16   373.7  985.13   395.7  980.42   403.2  979.43
   410.7  980.35   413.1  980.65     423   986.4   442.7 1003.91   482.2 1036.09
   561.2 1096.65   650.1 1162.15   689.6 1189.82   709.4 1203.08   808.2 1266.51
#Mann= 3 , 0 , 0
       0     .06       0   395.7    .045       0   410.7     .06       0
#XS Ineff= 2 , 0
          291.41  999.73
Permanent Ineff=
       F       F
Bank Sta=395.7,410.7
XS Rating Curve= 0 ,0
Exp/Cntr=0.3,0.1
